--- lmcrk.prj (project) ---

Proj Title=lmcrk
Current Plan=p01
Default Exp/Contr=0,0
English Units
Geom File=g01
Flow File=f01
Plan File=p01
BEGIN DESCRIPTION:
END DESCRIPTION:
DSS Export Rating Curves= 0
DSS Export Rating Curve Sorted= 0
DSS Export Volume Flow Curves= 0
DXF OffsetX= 0
DXF OffsetY= 0
DXF ScaleX= 0
DXF ScaleY= 0

--- lmcrk.p01 (plan) ---

Plan Title=Approximate Study - 100yr
Program Version=4.00
Geom File=g01
Flow File=f01
Subcritical Flow
K Sum by GR= 0
Std Step Tol= 0.01
Critical Tol= 0.01
Num of Std Step Trials= 20
Max Error Tol= 0.3
Flow Tol Ratio= 0.001
Split Flow NTrial= 30
Split Flow Tol= 0.02
Split Flow Ratio= 0.02
Log Output Level= 0
Friction Slope Method= 1
Unsteady Friction Slope Method= 2
Unsteady Bridges Friction Slope Method= 1
Parabolic Critical Depth
Global Vel Dist= 0 , 0 , 0
Global Log Level= 0
CheckData=True
Encroach Param=-1 ,0,0, 0
Run HTab= 0
Run UNet= 0
Run PostProcess= 0
Run WQNet= 0
UNET Theta= 0
UNET Theta Warmup= 0
UNET ZTol= 0
UNET ZSATol= 0
UNET MxIter= 0
UNET MaxInSteps= 0
UNET DtIC= 0
UNET DtMin= 0
UNET MaxCRTS= 0
UNET WFStab= 0
UNET SFStab= 0
UNET WFX= 1
UNET SFX= 1
UNET DSS MLevel= 1
UNET DZMax Abort= 0
UNET Convert EG Bridges= 0
UNET Use Existing IB Tables= 0
UNET Froude Reduction=False
UNET Froude Limit= 0
UNET Froude Power= 0
UNET Time Slicing=0,0, 5
Write IC File= 0
Echo Input=False
Echo Output=False
Write Detailed= 0
Detailed Automatic Start=False, 0
WQ ULTIMATE=-1
WQ Max Comp Step=1HOUR
WQ Output Interval=15MIN
WQ Output Selected Increments= 0
WQ Output face flow=0
WQ Output face velocity=0
WQ Output face area=0
WQ Output face dispersion=0
WQ Output cell volume=0
WQ Output cell surface area=0
WQ Output cell continuity=0
WQ Output face conc=0
WQ Output face dconc_dx=0
WQ Output face courant=0
WQ Output face peclet=0
WQ Output face adv mass=0
WQ Output face disp mass=0
WQ Output cell mass=0
WQ Output cell source sink temp=0
WQ Output cell source sink nsm=0
WQ Output MaxMinRange=-1
WQ Daily Max Min Mean=-1
WQ Daily Range=0
WQ Daily Time=0
WQ Create Restart=0
WQ Fixed Restart=0
WQ System Summary=False
Sorting and Armoring Iterations= 10
XS Update Threshold= 0.02
Hydraulics Update Threshold= 0.02
Energy Slope Method= 1
Volume Change Method= 0
XS Weighting Method= 0
Number of US Weighted Cross Sections= 1
Number of DS Weighted Cross Sections= 1
Upstream XS Weight=0.25
Main XS Weight=0.5
Downstream XS Weight=0.25
Number of DS XS's Weighted with US Boundary= 1
Upstream Boundary Weight= 1
Weight of XSs Associated with US Boundary= 0
Number of US XS's Weighted with DS Boundary= 1
Downstream Boundary Weight= 0.5
Weight of XSs Associated with DS Boundary= 0.5
Sediment Output Level= 4
Mass or Volume Output= 0
Output Increment Type= 1
Profile and TS Output Increment= 10
XS Output Flag= 0
XS Output Increment= 10
Disregard all LS=0
Disregard all Conn=0
Disregard all Breaches=0
Disregard all Pumps=0

--- lmcrk.f01 (steady flow) ---

Flow Title=USGS Regression Equation
Program Version=4.00
Number of Profiles= 1
Profile Names=P100yr
River Rch & RM=lmcrk,Main            ,16420.9
     493
River Rch & RM=lmcrk,Main            ,14973.9
     538
River Rch & RM=lmcrk,Main            ,13196.8
     595
River Rch & RM=lmcrk,Main            ,11900.9
     659
River Rch & RM=lmcrk,Main            ,9784
     717
River Rch & RM=lmcrk,Main            ,6808.5
     771
River Rch & RM=lmcrk,Main            ,6573.2
     985
River Rch & RM=lmcrk,Main            ,5623.7
    1043
River Rch & RM=lmcrk,Main            ,3830.3
    1102
River Rch & RM=lmcrk,Main            ,248.6
    1182
Boundary for River Rch & Prof#=lmcrk,Main            , 1
Up Type= 0
Dn Type= 3
Dn Slope=0.020656
DSS Import GetInterval= 0
DSS Import GetPeak= 0
DSS Import FillOption= 0

--- lmcrk.g01 (geometry) ---

Geom Title=USGS 3m DEM
Program Version=4.00

River Reach=lmcrk           ,Main
Reach XY= 30
     1680766.082      213466.916     1680857.491      212906.885
     1681123.788      212263.365     1681054.347       210262.85
     1680861.833      209787.305     1679994.486      209059.791
     1679915.007       208834.96     1680100.613      208218.608
     1680400.849      207694.011     1680422.546      207318.215
     1680501.965      207197.532     1680340.449       206505.24
     1680348.829      206135.766     1680092.644      205860.453
     1679955.754      205050.998     1680070.401      204702.969
     1680343.452      204406.594     1680600.833        204307.2
     1680692.923      204084.497     1680574.718      203947.374
     1680592.366      203634.999     1680209.846      203137.675
     1680037.079      202681.202     1680275.356      202018.257
     1680392.862      201318.822     1680411.144      200313.027
     1680316.092      200215.336     1680269.294      199794.809
     1679955.849      199276.053     1679601.523      199047.605

Type RM Length L Ch R = 1 ,16420.9 ,153,155.4,157.8
XS GIS Cut Line= 3
     1681221.159      213472.416     1680766.423      213456.922
     1680311.687      213441.428
#Sta/Elev= 30
    10.1    1232    50.6 1218.85   111.2 1194.96   161.8  1178.1     182 1167.72
   252.8 1138.62   262.9 1136.22     273 1136.19   293.2 1138.19   313.4 1142.13
   323.6 1141.55   343.8 1138.71   394.3 1135.48     450 1126.52     455  1125.9
     460  1126.5   465.1 1127.11   475.2 1133.43   485.3 1141.46   495.4 1145.22
   515.7 1151.19   535.9 1154.73   626.9 1158.75     728 1159.32   768.4 1163.59
   778.6 1166.76   808.9 1181.48   859.4 1211.19   869.6 1218.55     910 1235.12
#Mann= 3 , 0 , 0
       0     .06       0     450    .045       0     460     .08       0
Bank Sta=450,460
XS Rating Curve= 0 ,0
Exp/Cntr=0.3,0.1

Type RM Length L Ch R = 1 ,16265.5 ,135.6,135.2,134.9
XS GIS Cut Line= 2
     1681131.319      213356.719     1680464.224      213254.089
#Sta/Elev= 30
    10.1 1255.18    50.4 1236.61    80.6 1221.08    90.7 1213.72   100.7 1203.22
   171.3  1160.7   181.3 1151.88   211.5 1146.89   241.8 1146.42   312.3  1127.3
   347.6 1123.88   352.6 1123.35   357.6 1123.78   362.7 1124.21     413 1142.94
   433.2 1143.23   443.2 1146.27   453.3 1150.75   483.5 1167.17   493.6 1171.02
   533.9  1173.6   554.1 1178.07   564.1 1183.06   594.4 1202.52   614.5 1217.21
   624.6  1225.1   634.6 1235.18   644.7 1247.03   654.8 1255.44   674.9 1268.78
#Mann= 3 , 0 , 0
       0     .06       0   347.6    .045       0   357.6     .08       0
Bank Sta=347.6,357.6
XS Rating Curve= 0 ,0
Exp/Cntr=0.3,0.1

Type RM Length L Ch R = 1 ,16130.3 ,107.3,109.4,111.5
XS GIS Cut Line= 3
     1681134.393       213247.44      1681012.52      213197.729
     1680456.072       213122.36
#Sta/Elev= 30
    10.1 1256.94    30.4 1247.17    40.5 1238.72      81 1219.27   101.2 1206.64
   111.4 1196.44   121.5 1182.14   141.6 1165.53   151.7 1160.51   171.7 1157.03
   211.8  1154.2     282 1128.27   302.1 1123.86   347.2 1120.23   352.2 1120.13
   357.3 1120.68   392.3 1125.02   402.4  1128.3   422.4 1140.36   442.5 1160.02
   462.5 1172.91   492.6 1187.07   512.7 1200.45   572.8 1229.47   582.9 1235.92
   592.9 1244.93     653 1277.25   663.1 1283.29   673.1  1293.7   693.2 1304.83
#Mann= 3 , 0 , 0
       0     .06       0   347.2    .045       0   357.3     .08       0
Bank Sta=347.2,357.3
XS Rating Curve= 0 ,0
Exp/Cntr=0.3,0.1

Type RM Length L Ch R = 1 ,16020.9 ,210.6,212.5,214.5
XS GIS Cut Line= 3
     1681262.246      213168.643     1680820.033      213061.532
      1680377.82       212954.42
#Sta/Elev= 30
    10.1 1333.67    80.9 1291.77      91 1284.47   101.1 1273.88   171.9 1233.27
     182 1220.88   212.3 1192.61   232.6 1176.33   252.8 1164.52   313.4  1161.7
   323.6 1158.63   343.8 1145.45   384.2 1128.77   414.6 1121.12   449.9 1117.01
     455 1116.42   460.1 1116.51   495.4 1121.29   515.7 1129.66   566.2 1160.37
   576.3 1171.59   586.4 1179.28   647.1 1210.03   667.3  1225.5   717.9 1251.71
   738.1 1267.34   808.9 1301.94     819 1311.52   889.8 1346.66     910 1361.26
#Mann= 3 , 0 , 0
       0     .06       0   449.9    .045       0   460.1     .08       0
Bank Sta=449.9,460.1
XS Rating Curve= 0 ,0
Exp/Cntr=0.3,0.1

Type RM Length L Ch R = 1 ,15808.4 ,101.8,101.7,101.7
XS GIS Cut Line= 2
     1681225.397       212978.27     1680481.329      212719.557
#Sta/Elev= 30
    10.1 1278.39    70.7 1245.75   131.3 1183.02   141.4 1173.99   151.5 1168.57
   161.6 1166.77   222.2 1169.38   232.3 1165.51   242.4 1156.53   252.5 1151.09
   313.1 1129.27   333.3 1118.24   368.6 1113.38   373.7 1113.09   378.8 1114.13
     404 1120.51   444.4 1119.56   464.6 1121.89   474.7 1126.29   484.8 1134.42
   494.9  1146.1   525.2    1167   585.8 1196.53   646.4 1223.11   666.6 1236.54
   686.8 1246.11     707 1254.02   737.3 1259.42   747.4  1264.3   787.8 1267.36
#Mann= 3 , 0 , 0
       0     .06       0   368.6    .045       0   378.8     .08       0
Bank Sta=368.6,378.8
XS Rating Curve= 0 ,0
Exp/Cntr=0.3,0.1

Type RM Length L Ch R = 1 ,15706.7 ,84.2,85.8,87.3
XS GIS Cut Line= 3
     1681229.005      212905.875     1681087.889      212822.488
     1680558.702      212639.678
#Sta/Elev= 30
     9.6 1263.68    57.9  1238.1    67.5 1231.31    86.8 1212.12    96.4 1195.61
   115.7 1177.44   125.3 1171.29     135 1168.41   173.9  1168.9   193.9 1165.55
   253.9 1145.33   263.9 1141.24   273.9 1133.92   313.9 1117.89   348.8 1112.39
   353.9 1112.24     359 1113.54   383.9 1119.73   433.9 1119.08   453.8 1121.91
   483.8 1132.25   503.8 1143.42   523.8 1159.53   533.8 1162.76   593.8 1172.74
   603.8 1176.81   643.8 1185.93   663.8 1186.86   693.8 1197.17   723.8 1201.67
#Mann= 3 , 0 , 0
       0     .06       0   348.8    .045       0     359     .08       0
Bank Sta=348.8,359
XS Rating Curve= 0 ,0
Exp/Cntr=0.3,0.1

Type RM Length L Ch R = 1 ,15620.9 ,189.4,191.3,193.2
XS GIS Cut Line= 3
     1681361.086      212863.727     1680943.837      212682.265
     1680526.588      212500.804
#Sta/Elev= 30
    10.1 1316.22    60.7 1292.84    70.8 1287.71    80.9 1280.46   101.1 1272.77
   141.6 1253.49   171.9 1232.63   232.6 1176.21   242.7 1169.42   252.8 1167.82
   283.1  1168.7   293.2 1166.39   323.6 1155.96   353.9 1136.36   374.1 1121.79
   384.2 1116.12   394.3 1112.27   404.4 1110.41   424.7 1112.73   449.9 1110.46
     455 1109.99   460.1 1110.43   485.3 1115.84   495.4 1116.71   566.2 1118.43
   576.3  1120.8   677.4 1154.17     728 1167.77   758.3 1170.11     910 1209.42
#Mann= 3 , 0 , 0
       0     .06       0   449.9    .045       0   460.1     .08       0
Bank Sta=449.9,460.1
XS Rating Curve= 0 ,0
Exp/Cntr=0.3,0.1

Type RM Length L Ch R = 1 ,15429.6 ,214.1,208.7,203.4
XS GIS Cut Line= 3
     1681396.447      212678.933     1681240.364      212627.618
     1680767.838      212366.766
#Sta/Elev= 30
     9.7 1289.92    38.7 1277.85    48.3 1271.33    77.3 1257.35   106.3 1241.62
     116 1235.47   125.6 1226.08   174.3 1188.16   204.3  1170.1   214.3 1168.02
   234.3 1168.53   244.3 1167.46   254.3 1163.88   294.2 1141.95   304.2 1132.15
   334.2 1110.22  344.49 1107.19  387.79  1107.8  394.37 1106.93  401.67 1107.55
   424.2 1111.64   474.2 1112.51   484.2 1114.79   504.1 1127.54   574.1 1167.52
   584.1 1177.67   664.1 1225.03   674.1 1234.73   684.1 1241.95     704 1253.31
#Mann= 3 , 0 , 0
     9.7     .06       0  387.79    .045       0  401.67     .08       0
Bank Sta=387.79,401.67
XS Rating Curve= 0 ,0
Exp/Cntr=0.3,0.1

Type RM Length L Ch R = 1 ,15220.9 ,123.6,119.9,116
XS GIS Cut Line= 3
     1681552.789      212425.823     1681110.226      212320.176
     1680668.375       212211.53
#Sta/Elev= 30
    10.1 1172.37   111.2 1173.23   222.4 1169.47   242.7 1170.75     273 1169.91
   283.1 1168.31   303.3 1160.34   313.4 1150.67     364 1121.73   384.2 1108.59
   394.3 1104.45   449.8 1102.88     455  1102.5   460.2 1103.75   475.2  1108.2
   515.7 1108.59   525.8 1110.91   535.9 1115.55     546 1122.39   556.1 1131.53
   626.9 1169.04     637 1179.75   697.7 1218.02   707.8 1228.48   717.9 1236.38
   778.6 1271.95   798.8    1287   859.5  1314.9   879.7 1328.76     910 1342.44
#Mann= 3 , 0 , 0
       0     .06       0   449.8    .045       0   460.2     .08       0
Bank Sta=449.8,460.2
XS Rating Curve= 0 ,0
Exp/Cntr=0.3,0.1

Type RM Length L Ch R = 1 ,15101   ,126.2,127.1,128
XS GIS Cut Line= 5
      1681440.68      212328.581     1681312.392      212238.779
     1681256.266      212208.311     1680986.862      212195.482
     1680712.648      212153.789
#Sta/Elev= 30
     9.8    1140    39.1 1133.35     137 1120.05   165.7 1117.54   202.2 1115.66
   240.4 1121.89   260.4 1114.51   280.4 1104.11   290.4 1101.69   320.3 1103.37
   345.1 1099.14   350.3 1098.74   355.5 1099.15   380.3 1102.71   400.3 1112.22
   420.2 1125.98   460.2 1148.53   470.2 1157.48   480.2 1164.36   529.8 1193.55
   549.6 1211.86     609 1248.28   618.9 1255.34   628.8 1264.85   658.6 1280.16
   668.5 1286.54   698.2 1301.54   708.1 1310.72   757.6 1334.04   767.5 1339.98
#Mann= 3 , 0 , 0
     9.8     .06       0   345.1    .045       0   355.5     .08       0
#XS Ineff= 2 , 0
       0     320                       0
Permanent Ineff=
       F       F
Bank Sta=345.1,355.5
XS Rating Curve= 0 ,0
Exp/Cntr=0.3,0.1

Type RM Length L Ch R = 1 ,14973.9 ,184.9,182.7,179.8
XS GIS Cut Line= 2
     1681390.033        212099.5     1680823.429      212046.047
#Sta/Elev= 30
      10 1165.16    79.9 1129.12    89.9 1121.02    99.8 1116.14   139.8 1103.54
   149.8 1101.35   159.8 1100.61   189.7 1101.82   229.6 1100.95   244.4 1097.77
   249.6 1096.54   254.8 1096.93   259.6 1097.28   269.6 1099.97   279.6 1104.23
   299.5 1115.43   309.5  1122.9   329.5  1141.8   349.5 1153.59   369.4  1161.9
   389.4 1168.59   399.4 1174.45   429.3 1186.63   449.3 1196.46   469.3 1208.02
   479.3 1221.07   539.2 1264.54   549.2    1277   559.1 1284.56   569.1 1290.75
#Mann= 3 , 0 , 0
       0     .06       0   244.4    .045       0   254.8     .08       0
Bank Sta=244.4,254.8
XS Rating Curve= 0 ,0
Exp/Cntr=0.3,0.1

Type RM Length L Ch R = 1 ,14791.3 ,230.3,227.5,224.7
XS GIS Cut Line= 3
     1681603.703      211937.096       1681149.1      211922.739
     1680693.815      211911.458
#Sta/Elev= 30
    10.1 1288.13      91 1235.47   121.3 1232.08   151.6 1224.38   171.8  1226.1
     192 1218.93   232.5 1195.98   252.7 1177.83   303.2 1144.39   323.4 1123.63
   353.8 1102.66   363.9 1096.72   378.8 1093.79   384.1 1093.55   389.3 1094.28
   424.5 1097.46  452.56 1094.73     465  1100.3   535.8 1143.81     556 1161.87
   576.3 1173.45   606.6 1185.98   626.9  1201.6   687.6 1238.59   707.8 1257.26
   758.4 1287.58   778.7 1304.88   839.4 1336.99   859.7 1353.15   910.3 1376.51
#Mann= 3 , 0 , 0
    10.1     .06       0   378.8    .045       0   389.3     .08       0
Bank Sta=378.8,389.3
XS Rating Curve= 0 ,0
Exp/Cntr=0.3,0.1

Type RM Length L Ch R = 1 ,14563.7 ,190.2,189.5,188.8
XS GIS Cut Line= 2
     1681447.762      211682.566     1680812.739      211738.157
#Sta/Elev= 30
    10.1 1215.73    20.2 1207.88    30.4 1195.29   101.2 1143.64   111.3 1132.74
   141.7  1119.4     172 1108.23   182.1 1102.81   237.6  1089.3   242.8 1088.78
   248.1 1089.01     253 1089.21   263.1 1092.04   283.3 1093.33   303.5 1092.22
  310.05 1090.52   323.8 1095.79   333.9 1111.42   364.3 1132.22   404.7 1157.75
   414.8 1168.83   445.2 1186.24   475.6 1205.47   485.7 1218.02   556.5  1264.6
   566.6 1276.99   576.7  1284.2     597 1296.78   627.3 1311.89   637.5 1321.72
#Mann= 3 , 0 , 0
    10.1     .06       0   237.6    .045       0   248.1     .08       0
Bank Sta=237.6,248.1
XS Rating Curve= 0 ,0
Exp/Cntr=0.3,0.1

Type RM Length L Ch R = 1 ,14374.3 ,207.9,209.2,210.5
XS GIS Cut Line= 3
     1681570.938      211468.368     1681119.377      211524.205
     1680667.816      211580.043
#Sta/Elev= 30
    10.1  1252.5    70.8 1251.95      91 1247.99   101.1 1237.18   161.8 1206.18
   171.9 1195.86     182 1190.17   242.7 1162.55   262.9 1149.58     364  1107.9
   384.2 1091.68  391.79 1088.04   394.3  1087.1   404.4 1087.18   424.7 1089.74
  452.25 1088.23   465.1 1089.69   485.3 1108.54   535.9 1139.26   556.1 1157.63
   616.8 1195.65     637 1216.42   687.6 1249.76   707.8 1267.57     728 1276.84
   768.4 1288.92   788.7 1291.59   839.2 1284.39   859.4  1278.8     910 1270.14
#Mann= 3 , 0 , 0
    10.1     .06       0  391.79    .045       0   404.4     .08       0
Bank Sta=391.79,404.4
XS Rating Curve= 0 ,0
Exp/Cntr=0.3,0.1

Type RM Length L Ch R = 1 ,14165.1 ,212.8,213.4,214
XS GIS Cut Line= 2
      1681381.48      211297.703      1680663.07      211340.466
#Sta/Elev= 30
      10 1201.01      60 1166.74      70 1156.86      80  1148.8   139.9 1114.51
   159.9 1099.16   179.9 1087.66   194.6 1083.53   199.9 1083.02   209.9 1083.35
   249.9  1085.9   289.9 1084.04   299.9 1085.57   319.9 1092.56   359.8 1111.79
   369.8 1117.51   379.8 1126.63   449.8 1161.97   459.8 1171.85   479.8 1181.48
   489.8 1184.49   519.8 1185.21   599.7 1181.55   609.7 1179.73   619.7 1172.99
   629.7 1169.26   669.7 1158.05   689.7 1148.11   699.7 1144.56   719.7 1140.69
#Mann= 3 , 0 , 0
      10     .06       0   194.6    .045       0   209.9     .08       0
Bank Sta=194.6,209.9
XS Rating Curve= 0 ,0
Exp/Cntr=0.3,0.1

Type RM Length L Ch R = 1 ,13951.6 ,195.9,196.1,196.4
XS GIS Cut Line= 3
      1681543.31      211092.209     1680980.448      211105.038
     1680637.628      211167.442
#Sta/Elev= 30
    10.1 1323.22    20.1 1318.04    40.2 1302.34    90.5 1276.18   110.6 1260.84
   140.8 1248.31   160.9  1236.8   170.9 1230.04     191  1209.7   241.3 1175.86
   261.4 1156.11   321.7 1118.08   341.8 1099.43   361.9 1085.02   376.7 1079.94
     382 1079.36   387.4 1079.75   422.3 1082.77  468.58  1081.3   492.6 1086.05
   622.7 1103.65   682.5 1115.41   702.4 1121.23   712.3 1129.27   742.2 1143.03
   772.1 1152.69     792 1162.77   851.7 1183.56   871.6 1194.94   911.5 1209.47
#Mann= 3 , 0 , 0
    10.1     .06       0   376.7    .045       0   387.4     .08       0
Bank Sta=376.7,387.4
XS Rating Curve= 0 ,0
Exp/Cntr=0.3,0.1

Type RM Length L Ch R = 1 ,13755.5 ,185.8,184.8,183.9
XS GIS Cut Line= 2
     1681413.552       210902.15     1680641.688      210910.702
#Sta/Elev= 30
      10 1238.23    50.1 1214.92    70.2  1195.1   130.3 1156.59   150.4  1138.5
   200.5 1110.59   210.5 1104.25   230.6 1087.97   240.6 1081.32   250.6 1076.55
   255.2 1075.89   260.6 1075.11     266 1075.54   300.7 1079.64   330.8 1078.27
   360.9 1089.72   380.9 1093.44     421 1098.27   441.1 1104.05   451.1 1111.75
   511.3 1135.27   521.3 1142.24   531.3 1146.39   591.5 1168.31   601.5 1175.72
   671.7 1206.43   681.7 1215.02   741.8 1245.37   751.9 1253.88   771.9 1265.08
#Mann= 3 , 0 , 0
      10     .06       0   255.2    .045       0     266     .08       0
Bank Sta=255.2,266
XS Rating Curve= 0 ,0
Exp/Cntr=0.3,0.1

Type RM Length L Ch R = 1 ,13570.6 ,112.2,113.3,114.3
XS GIS Cut Line= 3
     1681534.118        210699.1     1681079.923      210726.156
     1680625.728      210753.212
#Sta/Elev= 30
    10.1 1190.86    40.4  1175.9    50.6 1168.36    60.7 1163.12   141.6  1141.3
   192.1 1131.24   212.3 1123.31     273 1105.22   293.2  1095.5   323.6 1085.08
   353.9 1072.64   358.6 1072.11     364  1071.5   369.4 1072.13   414.6 1075.98
     455 1073.51   465.1 1075.15   495.4 1085.77   576.3 1132.72   596.6 1152.01
   647.1 1184.56   667.3 1202.88   717.9 1225.97     728 1231.48   748.2 1245.29
   798.8 1267.67     819 1280.91   869.6 1300.74   889.8 1311.83     910 1318.58
#Mann= 3 , 0 , 0
       0     .06       0   358.6    .045       0   369.4     .08       0
Bank Sta=358.6,369.4
XS Rating Curve= 0 ,0
Exp/Cntr=0.3,0.1

Type RM Length L Ch R = 1 ,13457.4 ,69.6,69.1,68.6
XS GIS Cut Line= 4
     1681528.877      210630.374     1681275.509      210607.923
     1680913.097      210612.734     1680635.675      210712.157
#Sta/Elev= 30
     9.8  1172.2    39.1 1154.39    58.7 1147.65   107.6 1141.33   146.7 1126.48
   195.7  1112.8   215.2 1105.62   274.5 1090.59   294.6 1083.41   359.7 1068.53
   365.1 1067.12   370.6 1067.37   415.4 1073.36   455.7 1070.07   465.8  1071.2
   506.1 1088.79   516.1 1098.21   556.4 1120.13   586.6  1139.1   596.7 1152.25
   656.1 1188.98   675.7 1207.86   734.7 1247.01   744.5 1261.71   754.3    1271
   783.8 1291.41   823.1 1307.55   832.9 1315.01   872.2 1323.28   911.5 1337.18
#Mann= 3 , 0 , 0
       0     .06       0   359.7    .045       0   370.6     .08       0
Bank Sta=359.7,370.6
XS Rating Curve= 0 ,0
Exp/Cntr=0.3,0.1

Type RM Length L Ch R = 1 ,13388.2 ,193.5,191.4,189.4
XS GIS Cut Line= 3
     1681427.851      210532.554     1680868.196      210551.797
     1680648.504      210603.113
#Sta/Elev= 30
      10 1128.77      30 1121.78      40 1115.66      90 1102.72     120  1095.7
     180 1086.47     190 1083.64     250 1074.24     260 1072.16     270 1067.48
   274.5 1066.67     280 1065.69   285.4 1065.88     330 1070.46     360 1068.62
     370 1069.38     380  1072.9     410 1089.27     430 1104.82     480 1133.95
     500  1151.8     560 1189.53   569.8 1198.14   579.6 1209.18   638.5 1249.21
   648.3 1261.92   707.1  1304.7   726.7 1324.71   756.2 1343.06   785.6 1358.68
#Mann= 3 , 0 , 0
       0     .06       0   274.5    .045       0   285.4     .08       0
Bank Sta=274.5,285.4
XS Rating Curve= 0 ,0
Exp/Cntr=0.3,0.1

Type RM Length L Ch R = 1 ,13196.8 ,57.5,56.6,55.7
XS GIS Cut Line= 3
     1681352.482       210320.88     1680980.448      210372.195
     1680629.261      210434.735
#Sta/Elev= 30
     9.9 1189.93    49.4 1167.89    69.2 1151.93   118.6 1125.08   128.5 1118.86
   138.4 1109.03   197.7  1079.3   207.5 1072.79   247.1 1063.46   261.4 1061.19
   266.8 1060.72   272.3 1060.86   276.7 1060.97   306.4 1067.09   345.9 1067.32
   355.8 1074.22   365.7 1085.49     435 1127.75   444.9  1139.2   504.4 1174.77
   514.3 1184.38   524.2 1191.24   573.7  1219.8   583.6 1228.89   593.5 1240.26
   623.3 1263.44   662.9 1291.19   672.8 1300.87   712.5 1324.31   732.3 1339.64
#Mann= 3 , 0 , 0
       0      .1       0   261.4    .045       0   272.3      .1       0
Bank Sta=261.4,272.3
XS Rating Curve= 0 ,0
Exp/Cntr=0.3,0.1

Type RM Length L Ch R = 1 ,13140.2 ,131.5,131.6,131.6
XS GIS Cut Line= 3
     1681439.076      210235.889     1680964.412      210322.483
     1680703.026      210385.024
#Sta/Elev= 30
    10.1 1259.08    70.4 1221.55    80.4    1210    90.5 1203.16   140.7 1174.02
   150.8  1164.4   160.8 1157.07   221.1 1124.84   241.2 1109.56   291.5 1084.47
   311.6 1071.46   321.7 1068.44   366.4 1060.73   371.9 1060.26   377.4 1060.88
   422.2  1067.4   442.3 1065.67   452.3 1066.52   462.4 1078.64   472.4 1086.06
   492.5 1095.87   522.3 1112.65   542.2 1127.69     592 1154.17   631.8 1181.39
   681.6 1220.32   691.5 1236.17   701.5 1244.73   731.4 1267.99   751.3 1281.68
#Mann= 3 , 0 , 0
       0      .1       0   366.4    .045       0   377.4      .1       0
Bank Sta=366.4,377.4
XS Rating Curve= 0 ,0
Exp/Cntr=0.3,0.1

Type RM Length L Ch R = 1 ,13008.6 ,114,112.9,111.8
XS GIS Cut Line= 2
     1681387.895      210113.181     1680635.274      210247.883
#Sta/Elev= 30
    10.1 1242.14    30.2 1229.59    40.2 1217.82   100.6 1182.91   110.7 1173.24
   120.7 1167.18   181.1 1138.18   201.2 1125.06   251.5 1100.88   271.6 1086.62
   301.8  1071.8   311.9 1067.63   346.6 1058.76   352.1 1057.91   357.6 1058.11
   412.5 1063.21   442.7 1062.61   452.7 1064.86   482.9 1077.57     493 1085.95
   533.2 1105.91   563.4 1125.35   573.4 1138.61   583.5 1147.95   633.8 1189.64
   653.9 1214.17   684.1 1237.36   714.3    1258   734.4 1274.91   764.6 1289.44
#Mann= 3 , 0 , 0
       0      .1       0   346.6    .045       0   357.6      .1       0
Bank Sta=346.6,357.6
XS Rating Curve= 0 ,0
Exp/Cntr=0.3,0.1

Type RM Length L Ch R = 1 ,12895.8 ,224.3,215,204.3
XS GIS Cut Line= 4
      1681382.95      210024.215     1681134.393      210037.043
     1680855.368      210102.791     1680611.621       210160.52
#Sta/Elev= 30
      10 1256.58    29.9 1244.06    49.8 1227.04    99.6 1201.56   119.5 1186.36
   179.2  1157.4   189.2 1150.84   199.1 1141.29   258.8 1107.69   268.7 1096.68
   298.3 1079.41     328  1064.5   337.9  1061.3   357.6 1057.63   381.7 1056.13
   387.3 1056.06   392.8  1056.4   436.7 1061.44   476.2 1059.23   486.1  1062.4
     496 1072.94   505.9 1079.15   565.6 1111.47   585.7 1129.37   635.8 1164.48
   645.8 1173.19   655.8 1185.01   715.9 1225.69   725.9 1236.09     786 1268.74
#Mann= 3 , 0 , 0
       0      .1       0   381.7    .045       0   392.8      .1       0
Bank Sta=381.7,392.8
XS Rating Curve= 0 ,0
Exp/Cntr=0.3,0.1

Type RM Length L Ch R = 1 ,12680.8 ,173.3,167.6,163.2
XS GIS Cut Line= 4
     1681376.989      209951.748     1681042.988      209807.729
     1680834.521      209958.467     1680480.777      210113.148
#Sta/Elev= 30
    10.1 1274.45    40.4 1261.16    60.6 1246.59   111.1  1226.9   131.3 1213.12
     192 1185.43   222.3 1161.12   242.5 1150.41   272.8 1136.93     293 1132.25
   383.5 1092.75   403.3  1075.5   423.1 1064.06   452.8 1055.64   496.7 1052.07
   502.3 1052.01   507.8 1052.07   571.5 1057.49   601.2  1056.3     621 1061.43
   690.3 1107.12     720 1120.29   739.8  1136.8   799.2 1172.97     819 1188.64
   898.2  1232.8   937.8  1249.3   967.5 1247.37   977.4 1242.07  1007.1 1236.82
#Mann= 3 , 0 , 0
       0      .1       0   496.7    .045       0   507.8      .1       0
Bank Sta=496.7,507.8
XS Rating Curve= 0 ,0
Exp/Cntr=0.3,0.1

Type RM Length L Ch R = 1 ,12513.2 ,174.4,175.9,177.4
XS GIS Cut Line= 4
     1681159.115      209619.274     1680900.402      209659.898
     1680733.628      209895.092      1680492.02      210046.899
#Sta/Elev= 30
    10.1 1161.08     141 1146.26   191.4 1136.27   221.6 1123.92   241.7 1112.71
   261.9 1104.76   301.7 1084.99   321.5 1079.79   371.2 1054.02   385.5 1049.83
   391.1 1049.36   396.7 1049.89   440.8 1053.89   480.6 1054.37   500.5 1058.55
   540.3 1076.54   550.2 1078.38   569.9 1091.62   638.8 1130.42   648.6 1138.69
   658.4 1144.61   697.8  1166.7   707.6 1166.93   717.5 1171.65   737.2 1186.41
   776.5 1209.01   796.2 1212.94     806 1212.71   815.9 1209.06   835.5 1208.01
#Mann= 3 , 0 , 0
       0      .1       0   385.5    .045       0   396.7      .1       0
Bank Sta=385.5,396.7
XS Rating Curve= 0 ,0
Exp/Cntr=0.3,0.1

Type RM Length L Ch R = 1 ,12337.3 ,184,185.6,187.3
XS GIS Cut Line= 3
     1680978.448      209306.315     1680689.134      209658.251
     1680397.536      210010.521
#Sta/Elev= 30
    10.1 1312.99    91.1 1256.02   111.4 1245.52   121.5 1236.19   222.7 1161.79
     243 1152.62     324    1102   344.2  1087.3   354.3 1085.47   425.2 1056.17
   435.3    1050   445.5 1046.18     450 1045.97   455.6 1045.73   461.2 1046.53
   475.5 1049.32   515.2 1050.27   604.7 1058.06   614.7 1061.82   644.5 1077.08
   664.4 1090.86   704.1 1111.95   714.1 1116.55     724 1115.83   743.9 1125.34
   753.8 1128.71   843.3 1143.52   853.2 1141.16   873.1 1140.09   912.9 1147.47
#Mann= 3 , 0 , 0
       0      .1       0     450    .045       0   461.2      .1       0
Bank Sta=450,461.2
XS Rating Curve= 0 ,0
Exp/Cntr=0.3,0.1

Type RM Length L Ch R = 1 ,12151.7 ,113.1,110,107
XS GIS Cut Line= 2
     1680772.114      209311.383     1680316.693      209777.495
#Sta/Elev= 30
      10 1221.22    30.1 1207.51    40.1 1197.96    50.1 1189.23    70.2 1174.57
    80.2 1169.39    90.2 1165.51   120.3 1143.93   140.4 1125.59   190.5 1089.96
   200.5 1083.65   210.5 1079.03   220.6 1076.61   230.6 1070.03   240.6 1064.62
   260.7 1055.46   280.7 1045.07   285.1 1043.55   290.7 1041.61   296.4 1041.63
   300.8 1041.65   330.8 1046.11     391 1046.95   471.2 1050.59   521.3 1056.61
   541.4 1059.82   581.5 1062.81   601.5 1063.53   621.6 1065.44   651.7 1073.73
#Mann= 3 , 0 , 0
       0      .1       0   285.1    .045       0   296.4      .1       0
Bank Sta=285.1,296.4
XS Rating Curve= 0 ,0
Exp/Cntr=0.3,0.1

Type RM Length L Ch R = 1 ,12041.6 ,138.5,140.8,143
XS GIS Cut Line= 4
     1680743.116      209251.282     1680534.648      209381.173
     1680390.325      209581.623     1680204.308       209727.55
#Sta/Elev= 30
     9.8 1229.18    29.5 1218.58    68.8 1191.29    78.6 1183.69    88.4  1172.2
     167 1121.19   176.8 1112.09   186.7 1104.35   206.3 1096.64   245.6 1076.64
   265.4 1065.41   275.3 1058.84   304.9 1042.78   314.8 1039.94     319 1039.73
   324.7 1039.46   330.3 1039.61   374.1 1044.18   423.5 1044.08     463 1045.44
   482.7 1047.84   522.2 1055.13   571.4 1075.64   591.1 1086.03   610.8 1094.35
   640.4 1102.68   660.1 1109.33   669.9 1114.21   679.8 1121.28     729 1138.78
#Mann= 3 , 0 , 0
       0      .1       0     319    .045       0   330.3      .1       0
Bank Sta=319,330.3
XS Rating Curve= 0 ,0
Exp/Cntr=0.3,0.1

Type RM Length L Ch R = 1 ,11900.9 ,167.8,166.9,166
XS GIS Cut Line= 3
     1680687.116      209016.324     1680226.892      209525.196
     1680144.177      209746.763
#Sta/Elev= 30
    10.1  1286.5    40.4 1268.23    50.4 1266.62    70.6 1252.16   151.3 1201.19
   171.5 1185.98   191.7 1179.36   252.2 1141.19   272.4 1126.24   292.6 1114.66
   312.8 1108.15   353.1 1087.29   373.3 1073.27   393.5 1063.62   413.7 1054.95
   433.9 1049.49   458.5 1038.64   464.1 1037.53   469.8 1038.13   494.4 1040.67
   544.9 1040.93     565 1044.37   645.8 1077.15     676 1092.68   686.1 1100.64
   725.5 1121.89   784.7 1149.27   814.2 1159.96   873.3 1173.89   922.6 1171.93
#Mann= 3 , 0 , 0
       0      .1       0   458.5    .045       0   469.8     .06       0
Bank Sta=458.5,469.8
XS Rating Curve= 0 ,0
Exp/Cntr=0.3,0.1

Type RM Length L Ch R = 1 ,11733.9 ,137.4,138.7,140.1
XS GIS Cut Line= 3
     1680564.762      208878.903     1680143.763      209385.924
      1679971.51      209576.907
#Sta/Elev= 30
      10 1349.76    69.9 1306.05    79.9 1302.67    89.9 1295.99   109.8 1279.78
   129.8 1259.18   189.7 1213.52   209.7 1202.93   239.6  1174.8   289.6 1137.49
   319.5 1112.15   329.5 1106.54   349.5 1089.32   399.4 1067.54   449.3    1039
   463.6 1035.23   469.3 1035.17     475 1035.48   549.2 1038.05   579.1 1048.37
   639.1 1076.55   688.7 1103.39   708.5 1109.22     748 1130.33   767.8 1146.04
   807.4 1171.73   827.2 1179.47   837.1  1186.4   856.9 1200.42   916.2 1254.71
#Mann= 3 , 0 , 0
       0      .1       0   463.6    .045       0     475     .06       0
Bank Sta=463.6,475
XS Rating Curve= 0 ,0
Exp/Cntr=0.3,0.1

Type RM Length L Ch R = 1 ,11595.2 ,62.6,64.2,65.8
XS GIS Cut Line= 4
     1680436.829      208909.716     1680220.344      209086.112
     1680032.723      209284.958     1679938.111      209446.921
#Sta/Elev= 30
      10 1257.39    19.9 1249.16    29.9 1242.64    39.9 1231.97    59.8 1216.23
   119.7 1172.96   129.7 1162.41   159.6 1142.42   179.5 1134.47   189.5 1128.96
   209.4 1117.38   229.4 1102.24   289.4 1067.44   329.9 1048.99   350.1 1037.62
   360.3 1033.45   364.7 1033.25   370.4 1032.99   376.1  1033.4   451.4 1037.46
   461.5 1039.55   471.6 1043.49   512.1 1060.94   562.5 1088.97   582.3 1095.44
   631.6 1123.07   671.1 1149.36     681 1151.59   690.9 1155.73   740.2 1185.47
#Mann= 3 , 0 , 0
       0      .1       0   364.7    .045       0   376.1     .06       0
Bank Sta=364.7,376.1
XS Rating Curve= 0 ,0
Exp/Cntr=0.3,0.1

Type RM Length L Ch R = 1 ,11531   ,74.3,67.4,60.5
XS GIS Cut Line= 4
     1680407.965      208903.302     1680164.218      209060.454
     1680027.912      209183.931     1679883.589       209419.66
#Sta/Elev= 30
      10 1238.68      20 1228.35      30 1221.53      40 1217.89      80 1188.62
     100 1169.54     170 1128.53     180 1120.28     210 1106.83     240 1090.78
     250 1085.12     270 1069.61     352 1033.32   357.8 1031.43   363.5 1031.47
   396.5 1033.03   435.2 1039.66   454.6 1040.56   503.5 1057.49   552.9 1084.68
   562.8 1090.82   572.6 1099.62   592.4  1111.8   612.1 1119.64   651.6 1144.54
   681.2 1160.51     701 1176.54   710.8 1182.02   730.6  1189.3   750.3 1200.24
#Mann= 3 , 0 , 0
       0      .1       0     352    .045       0   363.5     .06       0
Bank Sta=352,363.5
XS Rating Curve= 0 ,0
Exp/Cntr=0.3,0.1

Type RM Length L Ch R = 1 ,11463.6 ,27.8,31.1,34.4
XS GIS Cut Line= 4
     1680388.721      208880.852     1680084.038      209025.175
     1680007.066       209174.31     1679784.166      209406.831
#Sta/Elev= 30
     9.9  1235.3    59.5 1198.98    69.4 1186.78    79.3  1179.9   138.8  1144.9
   148.7 1135.23   218.1 1099.92     238 1085.91   267.7 1071.41   307.4 1055.34
   317.3 1048.62   337.1 1042.46   356.9  1039.4   386.5 1027.85   390.6 1027.75
   396.4 1027.59   402.1  1029.3   455.6 1041.57   485.2 1042.31   495.1 1045.07
   525.1 1058.97   535.2 1061.26   545.2 1066.75   645.9 1135.29   655.9 1146.13
   746.5 1204.07   766.7 1223.57   786.8 1238.72   806.9 1249.67   827.1 1263.95
#Mann= 3 , 0 , 0
       0      .1       0   390.6    .045       0   402.1      .1       0
Bank Sta=390.6,402.1
XS Rating Curve= 0 ,0
Exp/Cntr=0.3,0.1

Type RM Length L Ch R = 1 ,11432.5 ,37.3,45.5,53.7
XS GIS Cut Line= 4
     1680376.895      208873.836     1680062.991      209021.768
     1679972.789      209151.659     1679755.101      209378.968
#Sta/Elev= 30
     9.9 1231.32    39.7 1209.31    59.5 1189.36    89.2 1168.19     119 1153.03
   138.8 1136.76   208.2 1101.66     228 1087.63   287.5 1058.94   307.4 1047.32
     347 1036.14   386.5 1029.65   400.6 1025.38   406.3 1024.43   412.1 1025.63
   426.1 1030.43     436 1030.62   455.7 1041.91   465.6 1044.68   495.3 1046.17
   554.3 1081.83     574 1090.41   593.7 1104.21   613.3 1123.87   672.4 1167.74
     692 1177.67   701.9 1185.17   711.7 1195.78   760.9 1230.54   819.9 1278.46
#Mann= 3 , 0 , 0
       0      .1       0   400.6    .045       0   412.1      .1       0
Bank Sta=400.6,412.1
XS Rating Curve= 0 ,0
Exp/Cntr=0.3,0.1

Type RM Length L Ch R = 1 ,11387   ,117.1,119.4,121.8
XS GIS Cut Line= 4
      1680365.87      208870.929     1680115.709      208982.112
     1679869.825       209121.09     1679711.603      209364.837
#Sta/Elev= 30
     9.8 1225.97    29.3 1211.68    48.9  1191.9      88 1164.08   107.5  1155.2
   127.1 1138.85   195.5  1103.9   215.1 1090.09     264 1066.59   293.9 1047.02
   334.3 1036.05   409.2 1023.02     415 1022.52   420.7 1023.44   435.2 1029.29
   455.3 1045.98   465.4 1049.87   505.8    1053   515.8 1055.59   525.9 1061.81
     536 1071.47   616.3 1128.26   636.4 1138.39   656.4 1157.55   726.5 1209.18
   746.6 1217.93   756.6 1225.22   786.7 1254.55   826.8 1287.39   846.8 1301.41
#Mann= 3 , 0 , 0
       0      .1       0   409.2    .045       0   420.7      .1       0
Bank Sta=409.2,420.7
XS Rating Curve= 0 ,0
Exp/Cntr=0.3,0.1

Type RM Length L Ch R = 1 ,11267.5 ,140.1,148.6,157.1
XS GIS Cut Line= 4
     1680342.351      208834.581     1680077.223      208890.172
     1679752.228      209029.151     1679581.178      209146.748
#Sta/Elev= 30
      10 1228.76    20.1 1220.34    30.1 1208.31    90.3 1166.65   100.3 1152.43
   120.4 1139.28   160.5 1117.76   190.6 1096.04   210.7 1086.25   240.8 1075.57
   260.9 1065.59   321.4 1043.05   331.5 1035.59   341.6  1031.4   406.5 1020.09
   412.3 1019.41   418.1 1019.78   452.7 1023.08   472.9  1027.5   513.3 1043.68
   553.7 1065.92   563.8 1069.71   634.2 1074.86   644.1 1078.34   663.9 1089.65
   673.8 1093.08   683.7  1093.9   723.2 1107.93   812.2 1131.62   831.9  1133.8
#Mann= 3 , 0 , 0
       0      .1       0   406.5    .045       0   418.1      .1       0
Bank Sta=406.5,418.1
XS Rating Curve= 0 ,0
Exp/Cntr=0.3,0.1

Type RM Length L Ch R = 1 ,11119   ,206,211.7,217.4
XS GIS Cut Line= 4
     1680433.811      208724.896     1680070.809      208806.786
     1679771.471      208800.371     1679474.004      208798.941
#Sta/Elev= 30
    10.1 1275.76    40.2  1258.1    50.3 1246.83   120.7    1208   130.7 1197.25
   191.1 1159.75   211.2 1142.68   261.5 1117.78   281.6 1104.05   311.8 1089.26
     352 1075.26     422 1043.04     432 1034.24     452 1025.83     516 1017.83
   521.8 1017.43   527.6 1017.51   601.7 1023.02   621.6  1027.1   651.6 1039.22
   671.5 1052.75   721.1 1076.27   740.9 1090.09   760.8 1098.83   780.6 1105.23
   820.3 1108.24     850 1125.16   889.7  1137.4   959.1 1143.72     969 1142.32
#Mann= 3 , 0 , 0
       0      .1       0     516    .045       0   527.6      .1       0
Bank Sta=516,527.6
XS Rating Curve= 0 ,0
Exp/Cntr=0.3,0.1

Type RM Length L Ch R = 1 ,10907.3 ,169.9,169.9,170
XS GIS Cut Line= 2
     1680250.411      208689.189     1679638.907      208496.757
#Sta/Elev= 30
      10 1144.51      20 1137.19    30.1 1126.82    90.2 1092.76   100.2 1083.74
   110.2 1077.36   170.3 1047.87   190.3 1034.05   210.4 1027.07   240.4 1019.58
   270.5 1015.98   304.7 1013.96   310.5 1013.93   316.4 1014.35   340.6 1018.45
   350.6 1023.13   370.6 1035.67   420.7  1061.3   430.7 1070.84   440.7 1076.99
   450.8 1084.92   470.8 1095.91   500.8 1114.76   520.9 1131.52   540.9 1134.14
   550.9 1136.73   560.9 1142.68     591 1165.43     601  1178.7   641.1  1209.8
#Mann= 3 , 0 , 0
       0     .08       0   304.7    .045       0   316.4      .1       0
Bank Sta=304.7,316.4
XS Rating Curve= 0 ,0
Exp/Cntr=0.3,0.1

Type RM Length L Ch R = 1 ,10737.3 ,79.7,79.6,79.5
XS GIS Cut Line= 3
     1680469.267      208551.565     1680162.748      208488.205
     1679591.267      208306.851
#Sta/Elev= 30
    10.1 1243.97    30.3 1225.03    90.9 1188.72   111.1  1171.4   171.6 1134.09
   191.8 1113.75     212 1100.69   262.5 1076.46     323 1057.23     343 1046.06
   402.9 1022.05   422.9 1015.42     447 1012.29   452.9 1011.95   458.8 1012.54
   472.9 1017.03   522.8 1047.82   572.8 1075.12   592.8 1090.93   662.7 1129.15
   672.7 1138.36   692.7  1150.1   712.7 1156.32   742.7 1153.84   752.7 1161.04
   762.7    1174   822.6 1218.38   842.6 1235.83   902.6 1273.21   912.6 1281.48
#Mann= 3 , 0 , 0
       0     .08       0     447    .045       0   458.8      .1       0
Bank Sta=447,458.8
XS Rating Curve= 0 ,0
Exp/Cntr=0.3,0.1

Type RM Length L Ch R = 1 ,10657.7 ,95.5,95.9,96.2
XS GIS Cut Line= 3
     1680411.172       208460.71     1680152.993      208401.377
     1679769.734      208281.107
#Sta/Elev= 30
     9.8 1184.79    49.1 1160.86    58.9 1150.75    98.1 1126.14   117.7 1115.87
   127.5 1108.04   137.4 1102.48   196.2 1075.88     206 1070.38   215.9 1063.15
     285 1035.98     295 1029.12   315.1 1020.35   335.2  1014.4   359.5 1011.34
   365.3 1010.87   371.2 1010.99   385.4 1012.85   395.5 1017.18   405.5 1024.28
   425.6  1041.8   435.6 1048.61   445.7 1053.36   455.7 1061.45     526 1095.72
   546.1 1111.08   616.4 1147.79   626.4 1158.16   636.5 1161.94   666.6 1160.62
#Mann= 3 , 0 , 0
       0     .08       0   359.5    .045       0   371.2      .1       0
Bank Sta=359.5,371.2
XS Rating Curve= 0 ,0
Exp/Cntr=0.3,0.1

Type RM Length L Ch R = 1 ,10561.9 ,87.1,88.5,89.9
XS GIS Cut Line= 3
     1680483.467       208413.37     1679801.405      208184.591
     1679645.321      208186.729
#Sta/Elev= 30
    10.1 1224.28    50.7 1196.86    60.8 1184.85   121.6 1148.29   141.9 1131.55
   202.7 1100.09   222.9 1085.67   263.4 1065.05   293.8 1052.02   314.1 1040.38
     385 1011.63   395.2  1008.7   419.7 1007.61   425.6 1007.56   431.5 1008.88
     456    1018   466.1 1023.94     537 1049.34   557.3  1063.9   618.1 1099.09
   628.2 1106.13   638.3  1118.5   709.3 1162.44   719.4 1167.12   748.7 1169.04
   758.4 1173.19   777.9 1186.73   797.5 1207.42   865.8 1251.47   875.5 1263.07
#Mann= 3 , 0 , 0
       0     .08       0   419.7    .045       0   431.5      .1       0
Bank Sta=419.7,431.5
XS Rating Curve= 0 ,0
Exp/Cntr=0.3,0.1

Type RM Length L Ch R = 1 ,10473.4 ,100.9,101.6,102.4
XS GIS Cut Line= 3
     1680480.126      208313.179     1680242.794      208250.639
     1679854.724      208088.676
#Sta/Elev= 30
     9.8 1189.71    39.3 1173.85    49.1 1167.01    68.7 1151.84   127.6 1118.96
   137.4 1109.72   147.3  1103.4   206.2 1073.91     216 1067.85   225.8 1060.18
   295.5 1030.88   315.5 1018.81   335.5 1010.77   345.6 1008.34   365.6 1005.15
   379.7 1004.37   385.6 1004.36   391.5 1005.81   405.6 1010.22   425.7 1017.55
   465.7 1034.74   475.7 1041.68   485.7 1045.91   545.8  1068.5   555.8 1073.46
   565.8 1080.03   595.9 1096.43   635.9 1120.06   655.9 1140.06   665.9 1146.94
#Mann= 3 , 0 , 0
       0     .08       0   379.7    .045       0   391.5      .1       0
Bank Sta=379.7,391.5
XS Rating Curve= 0 ,0
Exp/Cntr=0.3,0.1

Type RM Length L Ch R = 1 ,10371.7 ,128.6,128.9,129.3
XS GIS Cut Line= 3
     1680515.539      208229.492      1680361.46      208199.324
     1679766.526      207925.109
#Sta/Elev= 30
     9.8 1184.81    19.6 1178.88    29.4 1168.64    88.3 1136.56   117.8  1115.8
   167.1 1092.11   177.2 1086.32   187.2 1076.77   217.5 1060.13   257.8 1041.57
   277.9  1028.8   328.3 1007.29   362.7 1002.24   368.6 1001.93   374.6 1002.53
     409 1011.85   439.2 1017.31   519.8 1046.08   529.9 1053.29     540 1058.04
   590.4 1077.38   610.5 1086.96   620.6 1096.32   650.8  1111.5   691.2 1135.63
   701.2 1143.02   711.3 1155.38   761.7 1187.37   781.9 1194.87   812.1 1195.63
#Mann= 3 , 0 , 0
       0      .1       0   362.7    .045       0   374.6      .1       0
Bank Sta=362.7,374.6
XS Rating Curve= 0 ,0
Exp/Cntr=0.3,0.1

Type RM Length L Ch R = 1 ,10242.8 ,132.3,132.4,132.6
XS GIS Cut Line= 3
     1680515.405      208156.027     1680443.244      208099.901
     1679906.039      207841.722
#Sta/Elev= 30
     9.1 1164.03    36.6 1145.93    45.7 1136.97    73.1  1115.8    91.4 1107.65
   121.7 1085.96   131.8 1075.67     152 1063.54   182.3 1043.17   212.6 1028.89
   222.7 1022.83   263.2 1008.73   283.4  1003.7   317.8  998.72   323.8  998.66
   329.7  998.74   354.1 1000.42   384.4 1004.79   394.5 1007.66   404.6 1012.64
   434.9 1023.57   455.1 1032.41   475.3 1042.15   495.5 1056.98   566.2 1094.93
   586.4 1109.51     647 1140.98   657.1 1147.06   677.3 1162.53   687.4 1166.25
#Mann= 3 , 0 , 0
       0      .1       0   317.8    .045       0   329.7      .1       0
Bank Sta=317.8,329.7
XS Rating Curve= 0 ,0
Exp/Cntr=0.3,0.1

Type RM Length L Ch R = 1 ,10110.4 ,72.9,71.9,70.8
XS GIS Cut Line= 2
     1680633.136      208049.889      1679955.35      207714.203
#Sta/Elev= 30
    10.1 1098.47    60.5 1095.38    80.7 1095.88   110.9 1094.51     121 1090.59
   171.4 1062.73   191.6 1049.18   221.9 1031.54     242 1022.41   282.4 1008.84
   312.6 1000.67   357.1  996.91   363.1  996.85     369  996.92   393.3  997.17
   403.4  999.36   413.5  1005.8   423.6 1014.41   433.6 1021.53   443.7 1027.17
   453.8 1035.51   463.9 1041.88   615.2 1113.76   625.3 1122.08   655.5 1139.68
   685.8 1152.43   695.9 1158.25   705.9 1164.28     716 1174.81   756.4 1202.88
#Mann= 3 , 0 , 0
       0      .1       0   357.1    .045       0     369      .1       0
Bank Sta=357.1,369
XS Rating Curve= 0 ,0
Exp/Cntr=0.3,0.1

Type RM Length L Ch R = 1 ,10038.5 ,83.3,83.6,83.9
XS GIS Cut Line= 4
     1680696.612      208000.478     1680478.523      207883.416
     1680191.479      207759.939     1679989.426      207692.588
#Sta/Elev= 30
     9.9 1090.03    89.1 1078.99   138.6  1075.3   158.4 1070.69   168.3 1067.39
   178.2 1060.32   188.1 1054.94   217.8 1043.72   237.6    1034   257.6 1022.11
   267.7 1012.81   277.8 1006.35   287.8 1002.98   318.1  998.66   348.3  998.31
   368.5  996.15   412.9   995.8   418.9  995.56   424.8  996.52     429   997.2
   449.1 1011.24   489.4 1033.18   509.6 1042.87   529.8 1056.01   598.7 1087.33
   618.1 1101.04   685.8 1136.05   695.5 1145.08   734.3 1167.79     773  1192.1
#Mann= 3 , 0 , 0
       0      .1       0   412.9    .045       0   424.8      .1       0
Bank Sta=412.9,424.8
XS Rating Curve= 0 ,0
Exp/Cntr=0.3,0.1

Type RM Length L Ch R = 1 ,9954.9  ,178.4,170.9,163.5
XS GIS Cut Line= 3
     1680789.219      207936.568     1680267.516      207703.512
     1679972.455      207628.678
#Sta/Elev= 30
      10 1092.82    90.2 1082.32   100.2 1080.47   110.3 1077.04   180.4 1062.66
   210.5 1059.94   270.7 1037.77   290.7 1026.38   340.8 1006.22   350.9  1003.3
   380.9  998.61   445.1   993.3   451.1  992.94   457.1  993.01   471.1  994.62
   481.2  997.53   501.2  1004.9   531.3 1018.48   541.3 1027.21   610.7 1060.25
   620.5 1066.54   630.3 1074.37     699 1110.08   708.9  1119.4   767.8 1153.86
   797.2 1175.81   807.1 1181.39   836.5 1201.27     866 1227.44   875.8 1230.29
#Mann= 3 , 0 , 0
       0      .1       0   445.1    .045       0   457.1      .1       0
Bank Sta=445.1,457.1
XS Rating Curve= 0 ,0
Exp/Cntr=0.3,0.1

Type RM Length L Ch R = 1 ,9784    ,283.7,291.8,299.9
XS GIS Cut Line= 4
     1680819.153      207746.275     1680643.827      207600.882
     1680226.892      207579.501     1680021.632      207560.258
#Sta/Elev= 30
     9.9 1162.44    29.7 1159.91    49.5 1153.35    69.3 1150.42    79.2 1145.52
    89.1 1136.28   188.2 1088.88   198.1 1082.77     208 1073.65   227.8 1064.81
   267.5 1043.81   287.4 1029.47     347  1001.3   366.9  995.51   440.4   988.6
   446.4  988.46   452.5     989   506.1  999.14   535.9 1007.68   585.6 1032.31
   595.6 1041.18   605.5  1047.5   655.1 1073.65   674.7 1090.33   733.6 1124.23
   743.4 1131.82   753.2 1141.91   812.1 1179.55     822 1192.52   851.4  1213.2
#Mann= 3 , 0 , 0
       0      .1       0   440.4    .045       0   452.5      .1       0
Bank Sta=440.4,452.5
XS Rating Curve= 0 ,0
Exp/Cntr=0.3,0.1

Type RM Length L Ch R = 1 ,9492.1  ,286.2,276.4,266.5
XS GIS Cut Line= 4
     1680750.733      207588.054     1680468.895      207320.853
      1680342.67      207259.318     1679970.592      207298.184
#Sta/Elev= 30
       0 1135.49      10 1135.49    19.9 1128.64    49.8 1113.04    99.6 1082.35
   129.5 1067.05   139.4 1058.63     249 1013.06   298.7 1006.01   368.5  988.15
   428.5  983.62   438.5  983.32   448.5  984.94   458.6  989.19   528.8 1005.33
   538.9 1009.38     549 1015.49   599.6 1030.76   609.7 1035.82   619.8 1045.75
   629.9 1052.15   690.6 1081.76   700.7 1091.85   741.1 1115.81   761.3 1132.68
   771.5 1150.03     822  1189.1   842.2 1201.98   852.3 1212.24   902.9 1237.25
#Mann= 3 , 0 , 0
       0      .1       0   428.5    .045       0   448.5      .1       0
Bank Sta=428.5,448.5
XS Rating Curve= 0 ,0
Exp/Cntr=0.3,0.1

Type RM Length L Ch R = 1 ,9215.8  ,80.6,79.4,79
XS GIS Cut Line= 4
     1680921.086       207053.45     1680630.664      207064.981
     1680251.815      207075.805     1679965.344      207117.594
#Sta/Elev= 30
      10  1145.1    70.2 1136.64   140.3 1117.28   150.3 1113.57   160.4 1107.97
   190.4 1098.21   220.5 1086.77   230.5 1078.55   260.6 1062.88   280.6 1053.33
   300.6 1046.16   310.6 1040.13   370.4 1019.44   390.4 1009.49   450.2  989.49
   470.2  977.31   474.1  976.88   480.2  976.21   486.2  976.58     530  981.89
   579.9  984.26   599.8  986.84   609.8  989.62   669.7  1013.9   689.6 1024.56
   759.5 1049.95   769.5  1058.6   849.3 1093.88   919.2 1113.89   959.2 1122.39
#Mann= 3 , 0 , 0
       0      .1       0   474.1    .045       0   486.2      .1       0
Bank Sta=474.1,486.2
XS Rating Curve= 0 ,0
Exp/Cntr=0.3,0.1

Type RM Length L Ch R = 1 ,9136.3  ,172.3,172.5,181
XS GIS Cut Line= 3
     1680900.391       206950.19      1680442.69      206990.955
     1679988.133       207013.82
#Sta/Elev= 30
      10 1212.79    59.9 1191.02    69.9 1182.81   129.9 1156.07   139.9 1147.42
   209.8 1114.67   219.8  1105.8   229.8 1099.61   279.7 1072.64   289.7 1063.51
   299.7 1056.81   359.6 1030.56   379.6 1016.67   429.5  992.27   449.5  975.74
   453.4  975.15   459.5  974.24   465.6  974.54   550.5  983.56   661.8 1004.66
   671.9 1007.61     682 1012.09   732.6 1025.86   783.2 1046.94   813.5 1054.06
   833.7 1061.06   884.3  1074.5   894.4 1077.74   904.5  1082.6   914.6  1085.3
#Mann= 3 , 0 , 0
       0      .1       0   453.4    .045       0   465.6      .1       0
Bank Sta=453.4,465.6
XS Rating Curve= 0 ,0
Exp/Cntr=0.3,0.1

Type RM Length L Ch R = 1 ,8963.8  ,127.2,126.9,126.6
XS GIS Cut Line= 2
     1680725.075      206794.809     1680013.079      206858.952
#Sta/Elev= 30
    10.1 1183.04    20.1 1177.48    40.3 1163.18    60.4 1141.15    90.6 1120.53
   120.8 1102.12   130.9  1094.4     141 1085.18   191.3 1056.36   201.4 1048.66
   211.4 1038.14   271.9 1000.05   281.9  991.85     292  978.22   302.1  972.24
     306  971.66   312.1  970.75   318.3  971.19   422.9  979.25     433  981.38
     443  986.12   483.3  995.08   503.4 1000.49   513.5 1006.42   543.7 1016.82
     584 1032.12   594.1  1039.7   654.5 1065.19   664.5 1073.05   714.9 1097.09
#Mann= 3 , 0 , 0
       0      .1       0     306    .045       0   318.3      .1       0
Bank Sta=306,318.3
XS Rating Curve= 0 ,0
Exp/Cntr=0.3,0.1

Type RM Length L Ch R = 1 ,8837    ,87.6,87.2,86.9
XS GIS Cut Line= 4
     1680747.927      206687.134     1680518.613      206688.738
     1680205.912      206717.602     1680019.895      206767.314
#Sta/Elev= 30
      10 1210.37    19.9 1200.37    49.9 1181.81    69.8 1165.93    79.8 1157.45
    89.7 1142.94   139.6 1106.18   159.5 1094.34   169.5 1083.62   229.3 1050.99
   249.6 1033.74   290.1 1004.73   310.4  988.42   320.5  972.09   324.5  970.42
   330.6  967.87   336.8  968.17   431.9  972.48   452.2  974.24   462.3  976.53
   482.6  988.27   533.2 1008.44   543.4 1015.33   553.5 1020.25   614.3 1043.73
   634.6 1055.87   685.2 1076.64   695.4  1082.1   705.5 1090.41   735.9    1104
#Mann= 3 , 0 , 0
       0      .1       0   324.5    .045       0   336.8      .1       0
Bank Sta=324.5,336.8
XS Rating Curve= 0 ,0
Exp/Cntr=0.3,0.1
